--- BaldEagle.prj (project) ---

Proj Title=Bald Eagle Cr. for the WCDS Project
Current Plan=p01
Default Exp/Contr=0.3,0.1
English Units
Geom File=g01
Flow File=f02
Flow File=f01
Unsteady File=u02
Plan File=p01
Plan File=p02
Y Axis Title=Elevation
X Axis Title(PF)=Main Channel Distance
X Axis Title(XS)=Station
DSS Caption Additional Text=Jensen
BEGIN DESCRIPTION:
Bald Eagle Creek.  This model does not represent actual water surface elevations for Bald Eagle Creek.  This data set is intended to be used only as an example Unsteady Flow data set.
END DESCRIPTION:
DSS Start Date=02/18/99
DSS Start Time=0000
DSS End Date=02/21/99
DSS End Time=2400
DSS File=dss
DSS Export Rating Curves= 0
DSS Export Rating Curve Sorted= 0
DSS Export Volume Flow Curves= 0
DXF OffsetX= 0
DXF OffsetY= 0
DXF ScaleX= 1
DXF ScaleY= 10

--- BaldEagle.p01 (plan) ---

Plan Title=Unsteady with Bridges and Dam
Program Version=5.00
Short Identifier=UnsteadyFlow
Simulation Date=18FEB1999,0000,24FEB1999,0500
Geom File=g01
Flow File=u02
Subcritical Flow
K Sum by GR= 0
Std Step Tol= 0.01
Critical Tol= 0.01
Num of Std Step Trials= 20
Max Error Tol= 0.3
Flow Tol Ratio= 0.001
Split Flow NTrial= 30
Split Flow Tol= 0.02
Split Flow Ratio= 0.02
Log Output Level= 0
Friction Slope Method= 2
Unsteady Friction Slope Method= 2
Unsteady Bridges Friction Slope Method= 1
Parabolic Critical Depth
Global Vel Dist= 0 , 0 , 0
Global Log Level= 0
CheckData=True
Encroach Param=-1 ,0,0, 0
Computation Interval=2MIN
Output Interval=1HOUR
Instantaneous Interval=2HOUR
Mapping Interval=1HOUR
Run HTab= 1
Run UNet= 1
Run Sediment= 0
Run PostProcess= 1
Run WQNet= 0
Run RASMapper= 0
UNET Theta= 1
UNET Theta Warmup= 1
UNET ZTol= 0.01
UNET ZSATol= 0.1
UNET MxIter= 20
UNET Max Iter WO Improvement= 0
UNET MaxInSteps= 0
UNET DtIC= 0
UNET DtMin= 0
UNET MaxCRTS= 20
UNET WFStab= 2
UNET SFStab= 1
UNET WFX= 1
UNET SFX= 1
UNET DSS MLevel= 4
UNET Pardiso=0
UNET DZMax Abort= 100
UNET Use Existing IB Tables=-1
UNET Froude Reduction=False
UNET Froude Limit= 0.8
UNET Froude Power= 4
UNET Time Slicing=0,0, 5
UNET Junction Losses=0
UNET D1 Cores= 0
UNET D2 Coriolis=0
UNET D2 Cores= 0
UNET D2 Theta= 1
UNET D2 Theta Warmup= 1
UNET D2 Z Tol= 0.01
UNET D2 Max Iterations= 20
UNET D2 Equation= 0
UNET D2 RampUpFraction=0.5
UNET D2 TimeSlices= 1
UNET D2 BCVolumeCheck=0
UNET D1D2 MaxIter= 0
UNET D1D2 ZTol=0.01
UNET D1D2 QTol=0.1
UNET D1D2 MinQTol=1
DSS File=dss
Write IC File= 0
Write IC File at Fixed DateTime=0
Write IC File at Sim End=0
Echo Input=False
Echo Parameters=False
Echo Output=False
Write Detailed= 0
HDF Write Warmup=0
HDF Write Time Slices=0
HDF Flush=0
HDF Compression= 1
HDF Chunk Size= 1
HDF Spatial Parts= 1
HDF Use Max Rows=0
HDF Fixed Rows= 1
Stage Flow Hydrograph=Bald Eagle      ,Loc Hav         ,138154.4
Stage Flow Hydrograph=Bald Eagle      ,Loc Hav         ,137690.8
Stage Flow Hydrograph=Bald Eagle      ,Loc Hav         ,137327.0
Stage Flow Hydrograph=Bald Eagle      ,Loc Hav         ,136564.9
Stage Flow Hydrograph=Bald Eagle      ,Loc Hav         ,136202.3
Stage Flow Hydrograph=Bald Eagle      ,Loc Hav         ,135591.4
Stage Flow Hydrograph=Bald Eagle      ,Loc Hav         ,135068.7
Stage Flow Hydrograph=Bald Eagle      ,Loc Hav         ,134487.2
Stage Flow Hydrograph=Bald Eagle      ,Loc Hav         ,133881.0
Stage Flow Hydrograph=Bald Eagle      ,Loc Hav         ,133446.1
Stage Flow Hydrograph=Bald Eagle      ,Loc Hav         ,132973.6
Stage Flow Hydrograph=Bald Eagle      ,Loc Hav         ,132363.8
Stage Flow Hydrograph=Bald Eagle      ,Loc Hav         ,131699.7
Stage Flow Hydrograph=Bald Eagle      ,Loc Hav         ,130997.6
Stage Flow Hydrograph=Bald Eagle      ,Loc Hav         ,130339.2
Stage Flow Hydrograph=Bald Eagle      ,Loc Hav         ,129627.5
Stage Flow Hydrograph=Bald Eagle      ,Loc Hav         ,128760.7
Stage Flow Hydrograph=Bald Eagle      ,Loc Hav         ,128280.7
Stage Flow Hydrograph=Bald Eagle      ,Loc Hav         ,127410.9
Stage Flow Hydrograph=Bald Eagle      ,Loc Hav         ,126741.0
Stage Flow Hydrograph=Bald Eagle      ,Loc Hav         ,126454.1
Stage Flow Hydrograph=Bald Eagle      ,Loc Hav         ,126062.6
Stage Flow Hydrograph=Bald Eagle      ,Loc Hav         ,125704.7
Stage Flow Hydrograph=Bald Eagle      ,Loc Hav         ,125091.9
Stage Flow Hydrograph=Bald Eagle      ,Loc Hav         ,124615.5
Stage Flow Hydrograph=Bald Eagle      ,Loc Hav         ,124025.0
Stage Flow Hydrograph=Bald Eagle      ,Loc Hav         ,123503.5
Stage Flow Hydrograph=Bald Eagle      ,Loc Hav         ,123123.6
Stage Flow Hydrograph=Bald Eagle      ,Loc Hav         ,122703.3
Stage Flow Hydrograph=Bald Eagle      ,Loc Hav         ,122190.8
Stage Flow Hydrograph=Bald Eagle      ,Loc Hav         ,121754.0
Stage Flow Hydrograph=Bald Eagle      ,Loc Hav         ,121394.1
Stage Flow Hydrograph=Bald Eagle      ,Loc Hav         ,120862.6
Stage Flow Hydrograph=Bald Eagle      ,Loc Hav         ,120421.4
Stage Flow Hydrograph=Bald Eagle      ,Loc Hav         ,119954.9
Stage Flow Hydrograph=Bald Eagle      ,Loc Hav         ,119473.8
Stage Flow Hydrograph=Bald Eagle      ,Loc Hav         ,118901.0
Stage Flow Hydrograph=Bald Eagle      ,Loc Hav         ,118300.5
Stage Flow Hydrograph=Bald Eagle      ,Loc Hav         ,117753.9
Stage Flow Hydrograph=Bald Eagle      ,Loc Hav         ,117180.8
Stage Flow Hydrograph=Bald Eagle      ,Loc Hav         ,116401.3
Stage Flow Hydrograph=Bald Eagle      ,Loc Hav         ,115584.2
Stage Flow Hydrograph=Bald Eagle      ,Loc Hav         ,114899.8
Stage Flow Hydrograph=Bald Eagle      ,Loc Hav         ,113985.6
Stage Flow Hydrograph=Bald Eagle      ,Loc Hav         ,112856.9
Stage Flow Hydrograph=Bald Eagle      ,Loc Hav         ,111971.0
Stage Flow Hydrograph=Bald Eagle      ,Loc Hav         ,110657.4
Stage Flow Hydrograph=Bald Eagle      ,Loc Hav         ,109659.9
Stage Flow Hydrograph=Bald Eagle      ,Loc Hav         ,108600.1
Stage Flow Hydrograph=Bald Eagle      ,Loc Hav         ,107333.6
Stage Flow Hydrograph=Bald Eagle      ,Loc Hav         ,106466.0
Stage Flow Hydrograph=Bald Eagle      ,Loc Hav         ,105178.6
Stage Flow Hydrograph=Bald Eagle      ,Loc Hav         ,104647.2
Stage Flow Hydrograph=Bald Eagle      ,Loc Hav         ,104195.0
Stage Flow Hydrograph=Bald Eagle      ,Loc Hav         ,103854.0
Stage Flow Hydrograph=Bald Eagle      ,Loc Hav         ,103369.7
Stage Flow Hydrograph=Bald Eagle      ,Loc Hav         ,103122.3
Stage Flow Hydrograph=Bald Eagle      ,Loc Hav         ,101440.3
Stage Flow Hydrograph=Bald Eagle      ,Loc Hav         ,100657.3
Stage Flow Hydrograph=Bald Eagle      ,Loc Hav         ,99452.75
Stage Flow Hydrograph=Bald Eagle      ,Loc Hav         ,98206.87
Stage Flow Hydrograph=Bald Eagle      ,Loc Hav         ,97607.35
Stage Flow Hydrograph=Bald Eagle      ,Loc Hav         ,96370.43
Stage Flow Hydrograph=Bald Eagle      ,Loc Hav         ,94560.01
Stage Flow Hydrograph=Bald Eagle      ,Loc Hav         ,93391.71
Stage Flow Hydrograph=Bald Eagle      ,Loc Hav         ,92011.85
Stage Flow Hydrograph=Bald Eagle      ,Loc Hav         ,91030.01
Stage Flow Hydrograph=Bald Eagle      ,Loc Hav         ,90096.99
Stage Flow Hydrograph=Bald Eagle      ,Loc Hav         ,89060.69
Stage Flow Hydrograph=Bald Eagle      ,Loc Hav         ,87861.14
Stage Flow Hydrograph=Bald Eagle      ,Loc Hav         ,86942.04
Stage Flow Hydrograph=Bald Eagle      ,Loc Hav         ,85569.53
Stage Flow Hydrograph=Bald Eagle      ,Loc Hav         ,84724.08
Stage Flow Hydrograph=Bald Eagle      ,Loc Hav         ,83563.41
Stage Flow Hydrograph=Bald Eagle      ,Loc Hav         ,82607.89
Stage Flow Hydrograph=Bald Eagle      ,Loc Hav         ,81849.41
Stage Flow Hydrograph=Bald Eagle      ,Loc Hav         ,81084.18
Stage Flow Hydrograph=Bald Eagle      ,Loc Hav         ,80500.50
Stage Flow Hydrograph=Bald Eagle      ,Loc Hav         ,79684.28
Stage Flow Hydrograph=Bald Eagle      ,Loc Hav         ,78627.87
Stage Flow Hydrograph=Bald Eagle      ,Loc Hav         ,76643.40
Stage Flow Hydrograph=Bald Eagle      ,Loc Hav         ,76002.96
Stage Flow Hydrograph=Bald Eagle      ,Loc Hav         ,75917.82
Stage Flow Hydrograph=Bald Eagle      ,Loc Hav         ,75616.14
Stage Flow Hydrograph=Bald Eagle      ,Loc Hav         ,74650.60
Stage Flow Hydrograph=Bald Eagle      ,Loc Hav         ,74207.96
Stage Flow Hydrograph=Bald Eagle      ,Loc Hav         ,73504.24
Stage Flow Hydrograph=Bald Eagle      ,Loc Hav         ,72303.68
Stage Flow Hydrograph=Bald Eagle      ,Loc Hav         ,71400.81
Stage Flow Hydrograph=Bald Eagle      ,Loc Hav         ,70651.52
Stage Flow Hydrograph=Bald Eagle      ,Loc Hav         ,69567.33
Stage Flow Hydrograph=Bald Eagle      ,Loc Hav         ,68604.09
Stage Flow Hydrograph=Bald Eagle      ,Loc Hav         ,67326.78
Stage Flow Hydrograph=Bald Eagle      ,Loc Hav         ,66070.17
Stage Flow Hydrograph=Bald Eagle      ,Loc Hav         ,64908.02
Stage Flow Hydrograph=Bald Eagle      ,Loc Hav         ,63812.99
Stage Flow Hydrograph=Bald Eagle      ,Loc Hav         ,62746.41
Stage Flow Hydrograph=Bald Eagle      ,Loc Hav         ,61896.89
Stage Flow Hydrograph=Bald Eagle      ,Loc Hav         ,60901.09
Stage Flow Hydrograph=Bald Eagle      ,Loc Hav         ,59795.28
Stage Flow Hydrograph=Bald Eagle      ,Loc Hav         ,58836.23
Stage Flow Hydrograph=Bald Eagle      ,Loc Hav         ,58708.54
Stage Flow Hydrograph=Bald Eagle      ,Loc Hav         ,58091.91
Stage Flow Hydrograph=Bald Eagle      ,Loc Hav         ,57700.27
Stage Flow Hydrograph=Bald Eagle      ,Loc Hav         ,57250.60
Stage Flow Hydrograph=Bald Eagle      ,Loc Hav         ,56775.92
Stage Flow Hydrograph=Bald Eagle      ,Loc Hav         ,56243.79
Stage Flow Hydrograph=Bald Eagle      ,Loc Hav         ,55700.55
Stage Flow Hydrograph=Bald Eagle      ,Loc Hav         ,54696.51
Stage Flow Hydrograph=Bald Eagle      ,Loc Hav         ,53922.53
Stage Flow Hydrograph=Bald Eagle      ,Loc Hav         ,52879.19
Stage Flow Hydrograph=Bald Eagle      ,Loc Hav         ,51784.74
Stage Flow Hydrograph=Bald Eagle      ,Loc Hav         ,50720.68
Stage Flow Hydrograph=Bald Eagle      ,Loc Hav         ,49715.77
Stage Flow Hydrograph=Bald Eagle      ,Loc Hav         ,48965.94
Stage Flow Hydrograph=Bald Eagle      ,Loc Hav         ,48110.09
Stage Flow Hydrograph=Bald Eagle      ,Loc Hav         ,47453.14
Stage Flow Hydrograph=Bald Eagle      ,Loc Hav         ,46722.59
Stage Flow Hydrograph=Bald Eagle      ,Loc Hav         ,46310.48
Stage Flow Hydrograph=Bald Eagle      ,Loc Hav         ,45805.37
Stage Flow Hydrograph=Bald Eagle      ,Loc Hav         ,45233.89
Stage Flow Hydrograph=Bald Eagle      ,Loc Hav         ,44529.29
Stage Flow Hydrograph=Bald Eagle      ,Loc Hav         ,43919.30
Stage Flow Hydrograph=Bald Eagle      ,Loc Hav         ,42895.87
Stage Flow Hydrograph=Bald Eagle      ,Loc Hav         ,41806.43
Stage Flow Hydrograph=Bald Eagle      ,Loc Hav         ,40526.85
Stage Flow Hydrograph=Bald Eagle      ,Loc Hav         ,39499.37
Stage Flow Hydrograph=Bald Eagle      ,Loc Hav         ,38446.87
Stage Flow Hydrograph=Bald Eagle      ,Loc Hav         ,37962.54
Stage Flow Hydrograph=Bald Eagle      ,Loc Hav         ,37385.23
Stage Flow Hydrograph=Bald Eagle      ,Loc Hav         ,36769.88
Stage Flow Hydrograph=Bald Eagle      ,Loc Hav         ,36663.76
Stage Flow Hydrograph=Bald Eagle      ,Loc Hav         ,36339.56
Stage Flow Hydrograph=Bald Eagle      ,Loc Hav         ,35648.50
Stage Flow Hydrograph=Bald Eagle      ,Loc Hav         ,35072.37
Stage Flow Hydrograph=Bald Eagle      ,Loc Hav         ,34098.93
Stage Flow Hydrograph=Bald Eagle      ,Loc Hav         ,33498.68
Stage Flow Hydrograph=Bald Eagle      ,Loc Hav         ,32195.47
Stage Flow Hydrograph=Bald Eagle      ,Loc Hav         ,30878.12
Stage Flow Hydrograph=Bald Eagle      ,Loc Hav         ,29563.77
Stage Flow Hydrograph=Bald Eagle      ,Loc Hav         ,27226.40
Stage Flow Hydrograph=Bald Eagle      ,Loc Hav         ,25960.70
Stage Flow Hydrograph=Bald Eagle      ,Loc Hav         ,24843.25
Stage Flow Hydrograph=Bald Eagle      ,Loc Hav         ,24417.73
Stage Flow Hydrograph=Bald Eagle      ,Loc Hav         ,23872.06
Stage Flow Hydrograph=Bald Eagle      ,Loc Hav         ,23783.65
Stage Flow Hydrograph=Bald Eagle      ,Loc Hav         ,23384.79
Stage Flow Hydrograph=Bald Eagle      ,Loc Hav         ,22982.97
Stage Flow Hydrograph=Bald Eagle      ,Loc Hav         ,22386.15
Stage Flow Hydrograph=Bald Eagle      ,Loc Hav         ,21283.34
Stage Flow Hydrograph=Bald Eagle      ,Loc Hav         ,21199.93
Stage Flow Hydrograph=Bald Eagle      ,Loc Hav         ,20127.30
Stage Flow Hydrograph=Bald Eagle      ,Loc Hav         ,19036.24
Stage Flow Hydrograph=Bald Eagle      ,Loc Hav         ,18200.10
Stage Flow Hydrograph=Bald Eagle      ,Loc Hav         ,17549.23
Stage Flow Hydrograph=Bald Eagle      ,Loc Hav         ,16787.45
Stage Flow Hydrograph=Bald Eagle      ,Loc Hav         ,15407.88
Stage Flow Hydrograph=Bald Eagle      ,Loc Hav         ,14814.34
Stage Flow Hydrograph=Bald Eagle      ,Loc Hav         ,13326.74
Stage Flow Hydrograph=Bald Eagle      ,Loc Hav         ,12035.22
Stage Flow Hydrograph=Bald Eagle      ,Loc Hav         ,11865.80
Stage Flow Hydrograph=Bald Eagle      ,Loc Hav         ,11116.44
Stage Flow Hydrograph=Bald Eagle      ,Loc Hav         ,10995.73
Stage Flow Hydrograph=Bald Eagle      ,Loc Hav         ,10221.14
Stage Flow Hydrograph=Bald Eagle      ,Loc Hav         ,9258.941
Stage Flow Hydrograph=Bald Eagle      ,Loc Hav         ,8541.462
Stage Flow Hydrograph=Bald Eagle      ,Loc Hav         ,7936.130
Stage Flow Hydrograph=Bald Eagle      ,Loc Hav         ,6940.066
Stage Flow Hydrograph=Bald Eagle      ,Loc Hav         ,6267.489
Stage Flow Hydrograph=Bald Eagle      ,Loc Hav         ,5523.234
Stage Flow Hydrograph=Bald Eagle      ,Loc Hav         ,4293.710
Stage Flow Hydrograph=Bald Eagle      ,Loc Hav         ,3047.378
Stage Flow Hydrograph=Bald Eagle      ,Loc Hav         ,2731.142
Stage Flow Hydrograph=Bald Eagle      ,Loc Hav         ,2501.017
Stage Flow Hydrograph=Bald Eagle      ,Loc Hav         ,2371.827
Stage Flow Hydrograph=Bald Eagle      ,Loc Hav         ,1692.633
Stage Flow Hydrograph=Bald Eagle      ,Loc Hav         ,1212.855
Stage Flow Hydrograph=Bald Eagle      ,Loc Hav         ,659.942
Calibration Method= 0
Calibration Iterations= 20
Calibration Max Change=0.05
Calibration Tolerance=0.2
Calibration Maximum=1.5
Calibration Minimum=0.5
Calibration Optimization Method= 1
WQ AD Non Conservative
WQ ULTIMATE=-1
WQ Max Comp Step=1HOUR
WQ Output Interval=15MIN
WQ Output Selected Increments= 0
WQ Output face flow=0
WQ Output face velocity=0
WQ Output face area=0
WQ Output face dispersion=0
WQ Output cell volume=0
WQ Output cell surface area=0
WQ Output cell continuity=0
WQ Output cumulative cell continuity=0
WQ Output face conc=0
WQ Output face dconc_dx=0
WQ Output face courant=0
WQ Output face peclet=0
WQ Output face adv mass=0
WQ Output face disp mass=0
WQ Output cell mass=0
WQ Output cell source sink temp=0
WQ Output nsm pathways=0
WQ Output nsm derived pathways=0
WQ Output MaxMinRange=-1
WQ Daily Max Min Mean=-1
WQ Daily Range=0
WQ Daily Time=0
WQ Create Restart=0
WQ Fixed Restart=0
WQ System Summary=0
WQ Write To DSS=0
WQ Use Fixed Temperature=0
Sorting and Armoring Iterations= 10
XS Update Threshold= 0.02
Bed Roughness Predictor= 0
Hydraulics Update Threshold= 0.02
Energy Slope Method= 1
Volume Change Method= 1
Sediment Retention Method= 0
XS Weighting Method= 0
Number of US Weighted Cross Sections= 1
Number of DS Weighted Cross Sections= 1
Upstream XS Weight=0
Main XS Weight=1
Downstream XS Weight=0
Number of DS XS's Weighted with US Boundary= 1
Upstream Boundary Weight= 1
Weight of XSs Associated with US Boundary= 0
Number of US XS's Weighted with DS Boundary= 1
Downstream Boundary Weight= 0.5
Weight of XSs Associated with DS Boundary= 0.5
Sediment Output Level= 4
Mass or Volume Output= 0
Output Increment Type= 1
Profile and TS Output Increment= 10
XS Output Flag= 0
XS Output Increment= 10
Write Gradation File= 0
Read Gradation Hotstart= 0
Write HDF5 File= 0
Write DSS Sediment File= 0
SV Curve= 0
Specific Gage Flag= 0

--- BaldEagle.p02 (plan) ---

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Plan Title=Steady Flow Run
Version=Version 3.0 Beta April 15, 2000
Short Identifier=SteadyRun
Simulation Date=02/18/1999,0000,02/24/1999,0500
Geom File=g01
Flow File=f02
Friction Slope Method= 1
Global Vel Dist= 15 , 15 , 15
UNET MaxInSteps= 20
UNET Convert EG Bridges= 1
Write Velocity= 0
HTab Param Time=2/7/2000 3:55:25 PM
