HEC-RAS study BaldEagle.prj: Bald Eagle Cr. for the WCDS Project

--- BaldEagle.f02 (steady flow) ---

Flow Title=Steady Flow Data
Version=Version 3.0.0  Dec 2000
Number of Profiles= 8
Profile Names=.5 year,1 year,2 year,5 year,10 year,25 year,50 year,100 year
River Rch & RM=Bald Eagle,Loc Hav         ,138154.4
    2000    3000    5000   10000   15000   20000   25000   30000
Boundary for River Rch & Prof#=Bald Eagle,Loc Hav         , 1
Up Type= 0
Dn Type= 4
Dn Rating Curve # Pts= 7
       0   529.2    1000     535    3000     540   16500   557.3   27000   562.1
   32500   564.1   47000   568.6
Boundary for River Rch & Prof#=Bald Eagle,Loc Hav         , 2
Up Type= 0
Dn Type= 0
Boundary for River Rch & Prof#=Bald Eagle,Loc Hav         , 3
Up Type= 0
Dn Type= 0
Boundary for River Rch & Prof#=Bald Eagle,Loc Hav         , 4
Up Type= 0
Dn Type= 0
Boundary for River Rch & Prof#=Bald Eagle,Loc Hav         , 5
Up Type= 0
Dn Type= 0
Boundary for River Rch & Prof#=Bald Eagle,Loc Hav         , 6
Up Type= 0
Dn Type= 0
Boundary for River Rch & Prof#=Bald Eagle,Loc Hav         , 7
Up Type= 0
Dn Type= 0
Boundary for River Rch & Prof#=Bald Eagle,Loc Hav         , 8
Up Type= 0
Dn Type= 0
Gate Openings=Bald Eagle      ,Loc Hav         ,81500   ,Gate #1     ,
      10       1      10       1      10       1      10       1      10       1
      10       1      10       1      10       1
DSS Import GetInterval= 0
DSS Import GetPeak= 0
DSS Import FillOption= 0

--- BaldEagle.u02 (unsteady flow) ---

Flow Title=Flow Hydrograph 2
Program Version=6.30
Use Restart= 0
Initial Flow Loc=Bald Eagle      ,Loc Hav         ,138154.4,2000
Boundary Location=Bald Eagle      ,Loc Hav         ,138154.4,        ,                ,                ,                ,                                ,
Interval=1HOUR
Flow Hydrograph= 150
 1075.53 1301.64 1676.94 2199.12 2864.95 3670.34 4610.32 5679.08 6870.05 8175.88
 9588.5211099.2612698.7914377.2316124.2617929.0819780.5921667.3623577.75   25500
27422.2529332.6431219.4133070.9234875.7436622.7738301.2139900.7441411.4842824.12
44129.9545320.9246389.6847329.6648135.0548800.8849323.0649698.3649924.48   50000
49924.4849698.3649323.0648800.8848135.0547329.6646389.6845320.9244129.9542824.12
41411.4839900.7438301.2136622.7734875.7433070.9231219.4129332.6427422.2526133.62
24907.8423741.8422632.7121577.6720574.0819619.4518711.3617847.57 17025.916244.31
15500.8414793.62 14120.913480.9912872.2812293.2611742.4911218.57 10720.210246.14
  9795.2 9366.26 8958.23  8570.1  8200.9 7849.71 7515.65 7197.88  6895.6 6608.07
 6334.56 6074.39 5826.91  5591.5 5367.57 5154.56 4951.94  4759.2 4575.86 4401.47
 4235.58 4077.77 3927.67 3784.89 3649.07 3519.87 3396.97 3280.07 3168.87 3063.09
 2962.48 2866.76 2775.72 2689.12 2606.74 2528.38 2453.84 2382.93 2315.49 2251.33
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Stage Hydrograph TW Check=0
Use DSS=False
Use Fixed Start Time=False
Is Critical Boundary=False
Boundary Location=Bald Eagle      ,Loc Hav         ,81500   ,        ,                ,                ,                ,                                ,
Gate Name=Gate #1
Gate Use DSS=False
Gate Time Interval=1HOUR
Gate Use Fixed Start Time=False
Gate Openings= 150
       6    6.23    6.45    6.68     6.9    7.13    7.35    7.58     7.8    8.03
    8.25    8.48     8.7    8.93    9.15    9.38     9.6    9.83   10.05   10.28
    10.5   10.73   10.95   11.18    11.4   11.63   11.85   12.08    12.3   12.53
   12.75   12.98    13.2   13.43   13.65   13.88    14.1   14.33   14.55   14.78
      15   14.83   14.66   14.49   14.32   14.15   13.98   13.81   13.64   13.47
   13.31   13.14   12.97    12.8   12.63   12.46   12.29   12.12   11.95   11.78
   11.61   11.44   11.27    11.1   10.93   10.76   10.59   10.42   10.25   10.08
    9.92    9.75    9.58    9.41    9.24    9.07     8.9    8.73    8.56    8.39
    8.22    8.05    7.88    7.71    7.54    7.37     7.2    7.03    6.86    6.69
    6.53    6.36    6.19    6.02    5.85    5.68    5.51    5.34    5.17       5
       5       5       5       5       5       5       5       5       5       5
       5       5       5       5       5       5       5       5       5       5
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Boundary Location=Bald Eagle      ,Loc Hav         ,659.942 ,        ,                ,                ,                ,                                ,
Rating Curve= 7
   529.2       0     535    1000     540    3000   557.3   16500   562.1   27000
   564.1   32500   568.6   47000
Use DSS=False
Use Fixed Start Time=False
Is Critical Boundary=False
Precipitation Mode=Disable
Wind Mode=No Wind Forces
Air Density Mode=Specified
Met BC=Precipitation|Mode=None
Met BC=Precipitation|Expanded View=0
Met BC=Precipitation|Constant Units=mm/hr
Met BC=Precipitation|Point Interpolation=
Met BC=Precipitation|Gridded Source=DSS
Met BC=Evapotranspiration|Mode=None
Met BC=Evapotranspiration|Expanded View=0
Met BC=Evapotranspiration|Point Interpolation=Nearest
Met BC=Evapotranspiration|Gridded Source=DSS
Met BC=Wind Speed|Expanded View=0
Met BC=Wind Speed|Point Interpolation=Nearest
Met BC=Wind Speed|Gridded Source=DSS
Met BC=Wind Direction|Expanded View=0
Met BC=Wind Direction|Point Interpolation=Nearest
Met BC=Wind Direction|Gridded Source=DSS
Met BC=Wind Velocity X|Expanded View=0
Met BC=Wind Velocity X|Point Interpolation=Nearest
Met BC=Wind Velocity X|Gridded Source=DSS
Met BC=Wind Velocity Y|Expanded View=0
Met BC=Wind Velocity Y|Point Interpolation=Nearest
Met BC=Wind Velocity Y|Gridded Source=DSS
Met BC=Air Density|Mode=Constant
Met BC=Air Density|Expanded View=0
Met BC=Air Density|Constant Value=1.225
Met BC=Air Density|Constant Units=kg/m3
Met BC=Air Density|Point Interpolation=Nearest
Met BC=Air Density|Gridded Source=DSS
Met BC=Air Temperature|Expanded View=0
Met BC=Air Temperature|Point Interpolation=Nearest
Met BC=Air Temperature|Gridded Source=DSS
Met BC=Humidity|Expanded View=0
Met BC=Humidity|Point Interpolation=Nearest
Met BC=Humidity|Gridded Source=DSS
Met BC=Air Pressure|Mode=Constant
Met BC=Air Pressure|Expanded View=0
Met BC=Air Pressure|Constant Value=1013.2
Met BC=Air Pressure|Constant Units=mb
Met BC=Air Pressure|Point Interpolation=Inv Distance
Met BC=Air Pressure|Gridded Source=DSS
Non-Newtonian Method= 0 ,
Non-Newtonian Constant Vol Conc=0
Non-Newtonian Yield Method= 0 ,
Non-Newtonian Yield Coef=0, 0
User Yeild=   0
Non-Newtonian Sed Visc= 0 ,
Non-Newtonian Obrian B=0
User Viscosity=0
User Viscosity Ratio=0
Herschel-Bulkley Coef=0, 0
Clastic Method= 0 ,
Coulomb Phi=0
Voellmy X=0
Non-Newtonian Hindered FV= 0
Non-Newtonian FV K=0
Non-Newtonian ds=0
Non-Newtonian Max Cv=0
Non-Newtonian Bulking Method= 0 ,
Non-Newtonian High C Transport= 0 ,
Lava Activation= 0
Temperature=1300,15,,15,14,980
Heat Ballance=1,1200,0.5,1,70,0.95
Viscosity=1000,,,
Profile Coefficient=4,1.3,
Lava Param=,2500,

--- BaldEagle.g01 (geometry) ---

Geom Title=Existing Conditions - GIS Data
Program Version=3.10

River Reach=Bald Eagle      ,Loc Hav
Reach XY= 30
      1967609.38       288126.34        1969162.       290296.16
      1968887.13       292762.63      1970889.75       294943.97
      1972765.13       295643.84      1974573.75       294280.47
        1977661.        294589.5      1983420.38       301436.53
       1990774.5       307828.81      1992858.63       312472.09
       1994404.5       312918.47      1998621.63       312165.69
        2012330.       326268.47      2013869.38       327086.34
      2017013.13       325792.44       2020166.5       328480.91
       2024510.5       334273.81       2028609.5       334344.84
      2034689.63       338279.03        2037112.       340501.03
      2036252.13       343747.84      2037500.13       346710.75
      2039651.88       347285.81      2039689.25       349508.34
      2045787.13       347590.72       2047519.5       346142.34
      2055172.25       349196.34        2056631.         350650.
      2061241.13       350463.09      2065322.25       353446.47

Type RM Length L Ch R = 1 ,138154.4,358.43,463.64,517.64
XS GIS Cut Line= 2
      1968668.17       290166.79      1969067.87       289778.85
#Sta/Elev= 30
       0  660.41       5  660.61      40  659.85      90  658.45      95  658.48
     130   659.6     190  660.21     195  658.98     200   656.3     305  657.15
     310  657.68     320  660.58  324.99  661.39     330  660.95     345  658.84
     350  658.28     375  666.52     380  667.51     410  671.32     415  672.91
     430  678.12     440  683.19     445   685.6     455   688.7     460  689.95
     480   695.5     485  696.55  514.99  701.46     535  703.91  557.01  706.27
#Mann= 3 , 0 , 0
       0     .06       0     190     .04       0     375      .1       0
Bank Sta=190,375
XS Rating Curve= 0
Exp/Cntr=0.3,0.1

Type RM Length L Ch R = 1 ,137690.8,305.71,363.84,382.83
XS GIS Cut Line= 4
      1968627.02       290584.12      1969009.09       290343.13
      1969273.59       290290.23      1969408.78       290290.23
#Sta/Elev= 30
       0  664.28      55  661.54     160  658.65  180.01  658.79     250  658.98
  290.01  659.45     295  659.39     305  659.09     335  659.33     395  659.03
     450  659.45  460.01  660.06     465  660.27     510  659.64     520  659.96
     530  660.72     535  660.79     565  654.38     570  653.73     655  656.16
     660  658.06  672.56  664.59     705  681.46  721.46  689.01     735  694.24
     765  700.36     770  701.23     785  703.53     790  704.42  856.65   719.1
#Mann= 3 , 0 , 0
       0     .06       0     535     .04       0  672.56      .1       0
Bank Sta=535,672.56
XS Rating Curve= 0
Exp/Cntr=0.3,0.1

Type RM Length L Ch R = 1 ,137327.0,732.93,762.02,765.36
XS GIS Cut Line= 4
      1968585.88        290854.5      1968868.02       290736.95
       1969085.5       290672.29      1969391.15       290672.29
#Sta/Elev= 30
       0  662.72      20   665.5      25  666.48      65  664.33  254.99  658.93
     295  659.31     385  659.68     420  659.08     455  659.67     485  659.78
     515  659.58     520  659.38  524.99   658.8     530   658.5     550  658.12
     555  658.23     580   659.3     585  658.36     590  656.91     600  653.66
     605   653.4     705  656.01     710  659.27  717.24  663.79     745  681.14
     770  697.71     795   711.5     800  714.13     820  717.76  838.19  719.88
#Mann= 3 , 0 , 0
       0     .06       0     580     .04       0  717.24      .1       0
Bank Sta=580,717.24
XS Rating Curve= 0
Exp/Cntr=0.3,0.1

Type RM Length L Ch R = 1 ,136564.9,349.61,362.64,370.75
XS GIS Cut Line= 3
      1968521.22       291524.58      1968903.29       291424.66
      1969291.23       291430.54
#Sta/Elev= 28
       0  663.72      40  669.65      45  670.46   50.01  671.71      60  671.18
     210  666.85     265  663.38     270  662.78     340  659.16     420  658.46
     465  658.84     500  659.32  530.01  659.56  535.01  656.96     540  653.42
     675  655.83     680  657.03     685  659.22  700.46  667.61     715  675.36
     720  677.43     735  683.26     745   687.3     755  688.84     765  690.11
     775  691.22     780   691.6   782.9  691.71
#Mann= 3 , 0 , 0
       0     .06       0  530.01     .04       0  700.46      .1       0
Bank Sta=530.01,700.46
XS Rating Curve= 0
Exp/Cntr=0.3,0.1

Type RM Length L Ch R = 1 ,136202.3,590.5,610.86,647.38
XS GIS Cut Line= 3
      1968468.32        291918.4      1968715.19       291753.82
      1969255.96       291800.84
#Sta/Elev= 30
       0  657.88      20  657.23      35     659      50  659.66      95  657.17
     125  665.26     145  669.24     150  671.49     155  671.14     165  667.24
     200  656.24     205  655.79     245  657.12  285.01   656.5  330.01  657.03
     355  654.61     365  656.53     395  657.76     480  657.92     515  656.69
  539.89  657.03     545  656.56     550   654.3     555  653.47     690  654.75
     695  655.55  714.84  663.86     770  685.79     825  692.86  839.51  691.35
#Mann= 3 , 0 , 0
       0     .06       0  539.89     .04       0  714.84      .1       0
Bank Sta=539.89,714.84
XS Rating Curve= 0
Exp/Cntr=0.3,0.1

Type RM Length L Ch R = 1 ,135591.4,601.41,522.71,423.08
XS GIS Cut Line= 4
      1968485.96       292294.59      1968820.99       292335.73
      1969114.89        292423.9      1969355.88       292429.78
#Sta/Elev= 30
       0   658.4     170  657.21  194.99  659.81     225  655.88  268.29  657.66
     285  656.93  304.99  651.77  349.99  651.83  359.99  654.39  399.99  652.34
     440  653.81     445  652.07     505  654.78  529.99  652.84     560  666.11
     565   671.9  567.13  672.19  574.99  672.85     610  668.46  629.99  663.53
     650  656.73  689.99  655.43  699.99  652.34  754.99  652.34  764.99  656.19
  789.99  657.55  824.99  653.91  834.99  654.32     855  657.02  885.45  671.04
#Mann= 3 , 0 , 0
       0     .06       0  268.29     .04       0  567.13      .1       0
Levee=0,,,-1,574.99,,0,0
Bank Sta=268.29,567.13
XS Rating Curve= 0
Exp/Cntr=0.3,0.1

Type RM Length L Ch R = 1 ,135068.7,630.3,581.51,462.03
XS GIS Cut Line= 3
      1968177.37       293091.04      1969106.07       292785.39
      1969394.09       292814.78
#Sta/Elev= 30
       0  664.93  279.99   659.6     325  659.23  364.99  657.77     410  658.11
  509.99  654.55  689.99  654.33     730  654.93     740  656.09  749.99  652.93
  754.99  652.36     870  653.32  894.78  655.57  929.99  656.58 1029.99  654.52
 1044.99  652.01    1065  652.01    1070  652.75 1079.99  655.52 1149.99  656.41
 1174.99  656.53    1190  653.63    1205  653.63 1209.99  654.37    1215  658.01
    1220   662.8 1224.99  669.49 1234.99   673.1    1240  673.71 1267.22  670.33
#Mann= 3 , 0 , 0
       0     .06       0     740     .04       0  929.99      .1       0
Bank Sta=740,929.99
XS Rating Curve= 0
Exp/Cntr=0.3,0.1

Type RM Length L Ch R = 1 ,134487.2,605.29,606.25,590.87
XS GIS Cut Line= 3
       1968594.7       293702.34      1969164.85       293402.57
      1969564.55       293055.77
#Sta/Elev= 30
       0  669.08       5  669.03   24.99  661.37      75   661.8     170   658.5
  244.99  657.51  264.99  656.86  319.99  656.93  374.99  655.44     425  655.76
     480  654.73     640  655.43  679.99  654.99     730  655.66     750   651.2
  869.99  651.06  899.99  651.36  914.99  653.51  929.99  654.65    1015  655.69
 1034.99  656.93 1049.99  653.69    1055  653.37    1070   654.4 1094.99  657.01
 1124.99  657.17 1139.99  657.97    1160   670.7 1169.99  675.43 1173.33  675.19
#Mann= 3 , 0 , 0
       0     .06       0     730     .04       0  929.99      .1       0
Bank Sta=730,929.99
XS Rating Curve= 0
Exp/Cntr=0.3,0.1

Type RM Length L Ch R = 1 ,133881.0,465.19,434.84,425.17
XS GIS Cut Line= 3
      1969135.46       294207.84      1969670.35       293696.46
      1969993.63       293461.35
#Sta/Elev= 30
       0  665.68      20  658.03      25  656.71      75  653.65  120.01  654.39
     150  654.15     195   654.5     285  654.42     325  653.61     375  654.63
  475.01  653.48     560   653.8     655  652.94     715  652.94     735  652.76
     745  651.96     780  654.02     805  656.31  815.01  649.69     955   649.4
     970  652.56  990.01  653.56    1010  657.05    1030  652.89    1035  652.36
    1050   655.2    1100   660.6    1105  661.76    1135  673.88 1139.74  675.02
#Mann= 3 , 0 , 0
       0     .06       0     805     .04       0    1010      .1       0
Bank Sta=805,1010
XS Rating Curve= 0
Exp/Cntr=0.3,0.1

Type RM Length L Ch R = 1 ,133446.1,442.14,472.56,494.87
XS GIS Cut Line= 4
      1969546.91       294507.61      1969934.85       294043.26
      1970205.24       293825.78      1970287.53       293620.05
#Sta/Elev= 30
       0  664.63       5  664.98      25  660.23      45  653.36     110   652.7
     170   653.1  230.01  651.96     275  653.33     510  652.86     585  652.08
  625.01  651.21     705  653.21  726.26   650.1     735  648.51     740  648.49
     810  649.44     830  650.14     835  650.52  846.56  654.23     860  658.21
     865  657.41     880   653.5     885   653.1  905.01   656.7     935  666.13
  940.01  667.24    1005  670.53 1035.01  670.63 1100.01  672.09 1173.65  677.09
#Mann= 3 , 0 , 0
       0     .06       0  726.26     .04       0  846.56      .1       0
Bank Sta=726.26,846.56
XS Rating Curve= 0
Exp/Cntr=0.3,0.1

Type RM Length L Ch R = 1 ,132973.6,602.1,609.75,637.11
XS GIS Cut Line= 4
      1969843.75       294798.57      1970208.18       294410.63
      1970502.07       294199.02      1970784.21       293693.52
#Sta/Elev= 30
       0  660.19      50  659.73      80  666.13     110  664.97     120  662.94
     130  656.75     135   658.3     280  652.42     335  652.61     350  654.65
     405  650.96     435  653.43  532.27  652.99     550  649.95     570  649.95
  579.99  652.92     615  650.69     635  651.81     650  648.24  774.99  648.34
     790  651.53  822.11     652     990  653.11    1005  651.15    1025  655.37
    1095  654.48    1120  657.42    1135  654.22    1385  674.75 1473.32   672.7
#Mann= 3 , 0 , 0
       0     .06       0     635     .04       0  822.11      .1       0
Levee=-1,80,,0,,,0,0
Bank Sta=635,822.11
XS Rating Curve= 0
Exp/Cntr=0.3,0.1

Type RM Length L Ch R = 1 ,132363.8,749.24,664.14,507.86
XS GIS Cut Line= 5
      1970366.88       295115.97        1970602.       294845.59
       1970919.4       294645.74      1971225.05       294298.95
      1971336.73        293993.3
#Sta/Elev= 30
       0  753.43    9.99  742.53      40  720.86   79.99  686.96     115  665.13
  129.99  660.83     180   663.7     225  652.75     300  650.63     405  652.51
     450  646.86     470  647.93     490  645.25  569.99   646.8     590  653.22
     605  654.25  644.99  650.02     690  653.17     725  650.24  759.99  658.21
 1019.99  654.38    1040  657.64 1104.99  653.04    1130  660.26    1220  667.86
 1264.99  674.32 1324.99   675.9    1340  673.27 1419.99  669.64 1521.06  668.98
#Mann= 3 , 0 , 0
       0     .06       0     405     .04       0     605      .1       0
Bank Sta=405,605
XS Rating Curve= 0
Exp/Cntr=0.3,0.1

Type RM Length L Ch R = 1 ,131699.7,702.76,702.06,725.61
XS GIS Cut Line= 3
      1971113.37       295433.38      1971589.48       294522.31
      1971565.97       293958.03
#Sta/Elev= 30
       0  723.08      15  724.58      20  723.91      25  720.01      35   711.4
      50  695.21      80  660.09     110  659.57     135  663.69     165  662.68
     170  662.07     185  655.53     255  651.92     265  649.43     315  645.71
     375  647.88     425  647.52  449.15  652.86     790  652.19     860  654.05
     885  650.92    1045  650.21    1185  650.49    1245   651.5    1320  664.34
    1335  665.67    1380  668.11    1485  670.64    1555  673.98 1592.74  673.49
#Mann= 3 , 0 , 0
       0     .06       0     255     .04       0  449.15      .1       0
Bank Sta=255,449.15
XS Rating Curve= 0
Exp/Cntr=0.3,0.1

Type RM Length L Ch R = 1 ,130997.6,698.14,658.4,583.48
XS GIS Cut Line= 3
      1971777.57       295686.13      1972094.98       295027.81
      1972218.41       293758.18
#Sta/Elev= 30
       0  729.25   45.01  698.32   75.01  673.62      90  665.73      95  665.04
  110.01   665.4     155  654.19     220  649.74     235  644.98     380  645.49
     390  646.61     400  646.55     435   651.1     530  650.53     590  653.56
     595  653.46     615  650.69     650   651.5     815  650.58  870.01  649.44
    1065  650.26    1175  649.38    1440  649.82    1800  647.91    1845  648.55
    1870  650.11 1880.01   651.8    1915  654.81 1980.01  668.63 2006.46  668.89
#Mann= 3 , 0 , 0
       0     .06       0     220     .04       0     435      .1       0
Bank Sta=220,435
XS Rating Curve= 0
Exp/Cntr=0.3,0.1

Type RM Length L Ch R = 1 ,130339.2,753.78,711.7,428.92
XS GIS Cut Line= 3
      1972453.53       295991.78      1972735.67       294681.01
       1972647.5       293552.45
#Sta/Elev= 30
       0  659.66       5  660.36      10  665.65      15  664.59      20  658.82
      60  655.84      70  657.41     100  666.83     105  666.71     150  660.07
     180  651.88  270.28  649.85     280  649.44     300  642.94     305  642.71
     440     644     455  646.19     470  650.88     540   649.8     715  653.31
     990  648.15    2115   647.3    2235  649.17    2340  654.21    2370  659.96
    2380  666.44    2405  673.37 2415.01  674.06 2445.01  661.05 2472.79  661.54
#Mann= 3 , 0 , 0
       0     .06       0  270.28     .04       0     470      .1       0
Levee=-1,100,,0,,,0,0
Bank Sta=270.28,470
XS Rating Curve= 0
Exp/Cntr=0.3,0.1

Type RM Length L Ch R = 1 ,129627.5,792.27,866.78,581.35
XS GIS Cut Line= 5
      1973135.37       296256.28      1973252.92       295838.95
      1973211.78       295403.99      1973058.95       294681.01
       1972994.3        293540.7
#Sta/Elev= 30
       0  663.96   14.99   666.1      60  683.09   64.99  683.74      80  682.75
     115  677.21     170  652.41     185  649.11     300  650.84  449.99  650.64
  544.99  652.91  599.99  652.84  670.01  649.99  679.99  648.92     705  643.01
     795  642.66     910  644.52     985  647.55 1204.99   648.2 1289.99   646.7
    1460   646.4 2104.99   647.3    2370   645.7    2520  647.92 2634.99  654.07
 2664.99  670.37    2700  670.33 2709.99  667.01 2729.99  664.35 2751.57   665.4
#Mann= 3 , 0 , 0
       0     .06       0  670.01     .04       0     985      .1       0
Bank Sta=670.01,985
XS Rating Curve= 0
Exp/Cntr=0.3,0.1

Type RM Length L Ch R = 1 ,128760.7,690.64,480.04,527.21
XS GIS Cut Line= 5
       1974043.5       296329.76      1973996.48       295242.35
      1973490.98       294466.47      1973396.93       294078.53
      1973396.93       293543.64
#Sta/Elev= 30
       0  684.59     120  675.61     175  668.89     190  669.15     195   667.1
  210.01  653.85     215  652.41     290  646.55     580  646.56     615  648.02
  670.01  646.31    1050  645.66 1115.01  643.74 1200.01  645.97    1340  645.25
    1500  640.93 1565.01  642.43    1575  646.05 1850.01  646.09    1875  642.44
    1895  646.31    1970  644.43    2270  646.16 2590.01  644.27 2820.01  651.58
 2840.01  653.66 2880.01  669.36 2900.01   670.2 2920.01  661.83 2948.52  661.49
#Mann= 3 , 0 , 0
       0     .06       0    1340     .04       0    1575      .1       0
Bank Sta=1340,1575
XS Rating Curve= 0
Exp/Cntr=0.3,0.1

Type RM Length L Ch R = 1 ,128280.7,624.03,869.82,966.85
XS GIS Cut Line= 5
       1975001.6       296153.42      1974948.69       295765.48
      1973996.48       294384.18      1973867.16       294078.53
      1973826.02       293573.03
#Sta/Elev= 30
       0  665.64     140  659.94     165  657.62     250  653.87  259.99  652.23
     280  652.21     305  649.91     325  646.63     350  646.04     365  643.19
     415  641.89     485  643.72     565  643.02  724.99  644.67  904.99   644.7
    1240   642.9    1705  645.46    1785  643.08    1800  641.05    1900  641.52
 1909.99  644.98 1919.47  645.02    2490  643.12    2605  643.56    2710  645.28
    2790  649.41    2835  668.45    2865  668.79    2890  665.14 2908.29   665.5
#Mann= 3 , 0 , 0
       0     .06       0    1705     .04       0 1919.47      .1       0
Bank Sta=1705,1919.47
XS Rating Curve= 0
Exp/Cntr=0.3,0.1

Type RM Length L Ch R = 1 ,127410.9,525.47,669.85,687.62
XS GIS Cut Line= 4
      1975301.37       296088.76      1975342.51         295548.
      1974931.06       294566.39      1974837.01       293708.22
#Sta/Elev= 30
       0  662.35      75  660.83  194.99  651.49  309.99  648.42  399.99  651.22
  409.99  650.26  434.99   644.8  649.99  640.82  699.99  640.82  729.99  644.06
  774.99  640.73    1830  643.35 1869.99  639.31 1919.99  639.31    1970  641.09
    1985  639.37    2045   640.6    2050  641.56 2060.71  647.51 2074.99  654.17
 2104.99  652.36 2259.99  654.86 2304.99  653.53 2324.99  655.82 2344.99  663.44
 2349.99  664.14    2390  657.97    2400  655.13    2460  655.26 2469.99  657.49
#Mann= 3 , 0 , 0
       0     .06       0    1830     .04       0 2060.71      .1       0
Levee=0,,,-1,2349.99,,0,0
Bank Sta=1830,2060.71
XS Rating Curve= 0
Exp/Cntr=0.3,0.1

Type RM Length L Ch R = 1 ,126741.0,333.52,286.93,256.77
XS GIS Cut Line= 4
      1975868.58        295827.2      1975727.52       295333.46
       1975545.3       294751.54      1975533.54       293875.74
#Sta/Elev= 30
       0  660.64   55.01   656.8      85  656.06     150  657.08     255  654.91
  305.01  655.22     360  653.18     435  653.01     465  648.81     490  642.12
     500  641.81     645  640.52     700  641.79     755  640.27     875  639.38
    1155  640.27 1205.01  641.51 1315.01  641.18    1400   642.5    1410  638.23
    1415  637.54    1510  636.88    1515  636.99 1540.01  646.36 1554.14  647.87
    1675  650.12 1870.01  649.35    1915  661.54    1935   662.4 1999.16  656.61
#Mann= 3 , 0 , 0
       0     .06       0    1400     .04       0 1554.14      .1       0
Levee=0,,,-1,1935,,0,0
Bank Sta=1400,1554.14
XS Rating Curve= 0
Exp/Cntr=0.3,0.1

Type RM Length L Ch R = 1 ,126454.1,377.59,391.45,384.49
XS GIS Cut Line= 4
      1975986.14       295245.29      1975909.73       294916.13
      1975786.29       294140.24      1975792.17       293899.25
#Sta/Elev= 30
       0  673.87      15  674.98      45  679.61      95  680.88     120  685.88
  140.01  683.58     185  676.02     260   649.3     290  645.08     315   640.2
  337.91  637.82     390  637.44  430.01  639.05  455.01  638.79     505   640.2
     535  638.98     685     639     820  641.42     845  637.05     935  637.69
     945  640.88  962.47  641.98    1015  645.61    1060  646.56    1155   651.2
 1180.01  651.31    1260  660.08    1290  661.98 1310.01  659.34 1364.62  658.77
#Mann= 3 , 0 , 0
       0     .06       0     820     .04       0  962.47      .1       0
Bank Sta=820,962.47
XS Rating Curve= 0
Exp/Cntr=0.3,0.1

Type RM Length L Ch R = 1 ,126062.6,285.47,357.95,390.57
XS GIS Cut Line= 3
      1976238.89       295210.02      1976244.77        294498.8
      1976133.09       293934.52
#Sta/Elev= 30
       0   669.9      95  673.37     200  660.58     230  659.94     235  659.21
     260  645.19     275  638.25     305  639.36     320  642.23     345  637.14
     360  637.87     370  635.84     430   640.7     460   638.7     635  639.16
     800  641.12     825   639.6  865.28   639.4     885  635.25    1000  636.81
    1015  645.13    1020  645.99    1065  645.72    1095  648.01    1145  658.87
    1175  654.88    1180  654.82    1210  659.33    1255  656.29 1286.47  656.68
#Mann= 3 , 0 , 0
       0     .06       0  865.28     .04       0    1020      .1       0
Bank Sta=865.28,1020
XS Rating Curve= 0
Exp/Cntr=0.3,0.1

Type RM Length L Ch R = 1 ,125704.7,473.48,612.79,661
XS GIS Cut Line= 3
      1976485.76       295251.17      1976550.42       294345.97
      1976562.18       293987.42
#Sta/Elev= 30
       0  665.39   35.01   665.2     170  657.55  215.01  639.26  250.01  640.73
     260  643.48     265  643.81  295.01  637.13  350.01  636.54     370  635.58
     390  637.32  405.01   641.6  435.01  639.07     520  639.67  625.01  637.97
  880.01  638.64  963.74  641.64  970.01  640.74     990   635.5    1065   635.5
    1070  636.61 1095.01  652.46 1101.26  654.79 1135.01  654.53    1145  650.26
    1165  655.19    1195  660.46    1200  660.69 1245.01  654.78 1266.25  654.72
#Mann= 3 , 0 , 0
       0     .06       0  963.74     .04       0 1101.26      .1       0
Bank Sta=963.74,1101.26
XS Rating Curve= 0
Exp/Cntr=0.3,0.1

Type RM Length L Ch R = 1 ,125091.9,428.97,476.36,494.42
XS GIS Cut Line= 3
       1976662.1        295374.6      1976932.48       294904.37
      1977255.77        294099.1
#Sta/Elev= 30
       0  664.05      85  655.45     125  649.91  159.99  648.21     195  648.48
     220  640.04  259.99  642.69     305  636.39     380  638.02     510  636.75
     550  638.69     620  636.52     785  638.32     935  636.88 1014.99  639.72
 1039.99  634.55    1145  635.43    1150   637.6    1160  645.11 1172.97  647.46
    1200  649.29    1225  656.42    1235  657.43    1260  654.15    1310  658.78
    1325  661.87    1350  658.85    1375  664.54    1390  661.91 1410.16  663.42
#Mann= 3 , 0 , 0
       0     .06       0 1014.99     .04       0 1172.97      .1       0
Bank Sta=1014.99,1172.97
XS Rating Curve= 0
Exp/Cntr=0.3,0.1

Type RM Length L Ch R = 1 ,124615.5,441.73,914.18,662.11
XS GIS Cut Line= 3
      1976859.01       295589.14      1977323.36       295001.35
      1977693.67       294366.54
#Sta/Elev= 30
       0  664.71      80  654.66  134.99  650.12     210  646.25     235  641.75
     320  637.44     385  637.18  434.99  638.91     455  637.16     485  638.71
     505  636.65  549.99  637.32     575  635.08     595  636.76  834.99  638.19
     865  633.94  929.99  637.34     985  635.89    1030   639.3    1085  636.93
 1109.14  637.84    1205  633.44    1255  633.03 1319.99  635.37 1339.99  648.04
  1354.6  653.12    1360  654.93 1424.99  660.09 1469.99  654.88    1484  656.96
#Mann= 3 , 0 , 0
       0     .06       0 1109.14     .04       0  1354.6      .1       0
Bank Sta=1109.14,1354.6
XS Rating Curve= 0
Exp/Cntr=0.3,0.1

Type RM Length L Ch R = 1 ,124025.0,572.63,521.51,485.35
XS GIS Cut Line= 3
      1977035.35        295812.5      1977834.74       295048.38
      1978228.56       294848.53
#Sta/Elev= 30
       0  664.32     105  654.95  209.99  648.91     265   643.4  374.99  637.59
     470  637.13  489.99  635.23     540  636.31  559.99  639.53     620  638.59
     645  635.21  684.99  636.43  759.99  636.03     785  634.48  799.99  638.78
 1024.99  636.24    1060  633.82    1080  635.91 1214.99  637.73 1234.99  633.82
 1344.99  634.05 1349.99  635.19 1387.62  655.85    1410  656.38    1445  662.18
 1469.99   658.9 1509.99  671.11 1514.99  671.01 1524.99  667.61 1547.48  668.98
#Mann= 3 , 0 , 0
       0     .06       0 1214.99     .04       0 1387.62      .1       0
Bank Sta=1214.99,1387.62
XS Rating Curve= 0
Exp/Cntr=0.3,0.1

Type RM Length L Ch R = 1 ,123503.5,421.82,379.84,377.71
XS GIS Cut Line= 2
      1977382.14       296218.08       1978563.6       295154.18
#Sta/Elev= 30
       0  663.98      60  654.91     130  649.74     240  643.58  330.01  641.44
     385   635.8  645.01  638.04     720  637.18     745  633.47     765  637.68
     820  636.68     875   637.8     900  634.11     960  636.58    1065  634.18
    1165  635.77    1195  632.59    1310  631.32 1324.06  639.31    1360  648.61
    1390   653.1    1405  656.88    1430  655.91    1470  662.38    1495  658.69
    1515   666.6    1535  672.39 1545.01  670.57    1560  664.78 1589.88  666.85
#Mann= 3 , 0 , 0
       0     .06       0    1165     .04       0 1324.06      .1       0
Bank Sta=1165,1324.06
XS Rating Curve= 0
Exp/Cntr=0.3,0.1

Type RM Length L Ch R = 1 ,123123.6,443.87,420.36,415.79
XS GIS Cut Line= 2
      1977752.45       296435.56      1978869.25       295371.66
#Sta/Elev= 30
       0  663.06      30  655.46      95  648.19     175  642.46     245   640.5
     315  634.25     630  637.01     670   635.4     695  636.73     715  633.66
     730  636.52     770  633.74     800  635.94     885  633.91     965   636.3
  989.99   633.2    1005     636    1055   632.6    1070  630.09    1205  630.46
 1230.87  636.98    1260  641.02    1295  650.42    1305   655.7    1355  662.31
 1394.99  657.99    1420  660.17    1430  662.73    1460  662.53 1542.44  668.33
#Mann= 3 , 0 , 0
       0     .06       0    1005     .04       0 1230.87      .1       0
Bank Sta=1005,1230.87
XS Rating Curve= 0
Exp/Cntr=0.3,0.1

Type RM Length L Ch R = 1 ,122703.3,487.95,512.48,505.87
XS GIS Cut Line= 2
       1978043.4       296779.42      1979166.08       295650.86
#Sta/Elev= 30
       0  665.39      15  665.01   55.01  654.62  100.01  646.94  205.01  642.39
     260  637.81     335  639.31     390  635.72     405  632.96  490.01  633.19
  655.01  635.99     715  635.78  765.01  633.98     945  633.03    1135  634.47
 1155.01  629.92 1285.01  630.46 1300.01  638.19    1315  646.84 1330.01  654.19
    1335   655.5    1365  656.93 1390.01  661.63    1430  660.37 1450.01  666.36
    1470  669.65 1485.01  669.28    1510  664.44    1535  662.36 1591.87  665.98
#Mann= 3 , 0 , 0
       0     .06       0    1135     .04       0 1300.01      .1       0
Bank Sta=1135,1300.01
XS Rating Curve= 0
Exp/Cntr=0.3,0.1

Type RM Length L Ch R = 1 ,122190.8,423.09,436.79,441.86
XS GIS Cut Line= 2
      1978357.87       297099.76       1979545.2        296000.6
#Sta/Elev= 30
       0  663.72      80  646.87     135   642.4     290  637.63     370  637.89
     470  634.04  564.99  633.19  669.99  634.59     820  632.91     890  635.21
  969.99  632.63    1050  634.73    1065  631.04 1149.99  629.07    1175   633.4
    1190  629.05    1265  630.33 1283.23  640.53 1300.01  650.76    1315  653.88
    1335  655.75 1360.01  653.37    1375  658.31    1400  663.02 1424.99  662.08
    1450  665.25    1485  676.61    1535  666.35    1585  662.23 1617.99  663.36
#Mann= 3 , 0 , 0
       0     .06       0    1050     .04       0 1283.23      .1       0
Bank Sta=1050,1283.23
XS Rating Curve= 0
Exp/Cntr=0.3,0.1

Type RM Length L Ch R = 1 ,121754.0,361.03,359.88,359.74
XS GIS Cut Line= 2
      1978660.58       297349.57      1979906.69       296285.67
#Sta/Elev= 30
       0  672.86      30  665.49      85  649.33     115  642.85  160.01  639.41
     260  636.97     365  636.39     385  634.35  410.01  636.45     440  632.96
     790  631.77     840  629.76    1020  634.34    1035  629.34    1045  627.93
    1190  630.12    1200  631.52 1223.63  641.38    1250  648.87    1280  653.81
    1320   652.7 1344.99  658.83    1380  662.15    1390  661.01 1404.99   661.9
    1450  673.46    1475  675.84    1515  668.51    1590   662.3  1638.5  663.56
#Mann= 3 , 0 , 0
       0     .06       0    1020     .04       0 1223.63      .1       0
Bank Sta=1020,1223.63
XS Rating Curve= 0
Exp/Cntr=0.3,0.1

Type RM Length L Ch R = 1 ,121394.1,462.9,531.56,619.74
XS GIS Cut Line= 2
      1978977.99        297555.3      1980159.44       296538.42
#Sta/Elev= 30
       0  680.61      10  678.89      45  667.37      80  651.84     135  638.97
     165  638.37     225  634.05     275  635.13     295  632.07     340  633.01
     490  631.39     585  632.47     810  629.45  945.01  633.72     950  633.25
  964.99  628.28     985   627.2    1130  628.92  1151.8  639.87    1170  645.96
    1195  650.61    1300  663.52    1310  661.77    1330  662.34    1365   670.6
    1405  674.26    1425  674.78    1450  669.82    1545  662.02  1558.8  662.16
#Mann= 3 , 0 , 0
       0     .06       0  945.01     .04       0  1151.8      .1       0
Bank Sta=945.01,1151.8
XS Rating Curve= 0
Exp/Cntr=0.3,0.1

Type RM Length L Ch R = 1 ,120862.6,506.39,441.14,441.89
XS GIS Cut Line= 3
      1979260.13       297960.87      1979700.97       297484.76
      1980653.19       297020.41
#Sta/Elev= 30
       0  687.39      45  680.89   54.99  677.17      65  669.91      95   663.5
     160  640.91     215  635.98  309.99  632.82  444.99  634.59  479.99   632.2
     650  632.42  884.99   628.7  997.46  632.42    1010  629.11    1050  627.45
    1145  628.02    1155  631.34    1180  632.18 1214.07   645.2 1224.99  650.63
    1295  656.12    1330     652    1360  651.61    1380  659.03    1400  661.19
 1454.99  659.54    1485  668.09    1525  672.82    1595  674.07 1708.27  665.16
#Mann= 3 , 0 , 0
       0     .06       0  997.46     .04       0 1214.07      .1       0
Bank Sta=997.46,1214.07
XS Rating Curve= 0
Exp/Cntr=0.3,0.1

Type RM Length L Ch R = 1 ,120421.4,459.43,466.56,457
XS GIS Cut Line= 3
      1979601.04       298237.13      1980188.83       297737.51
      1980952.96       297331.94
#Sta/Elev= 30
       0  685.46      40  678.61      85  660.12  120.01  642.58     135  642.48
     155  636.99     395  633.72     425  630.69  460.01  633.11     500  630.53
     685  630.62     715  626.56  770.01  626.97     795  630.85  849.03  631.65
     885  626.96     980  627.61 1004.83  643.05 1020.01  645.93    1220  663.15
    1265  662.35    1300  655.39    1320  656.54    1365  664.21    1395  661.74
    1450  681.06    1475  684.44    1565   679.6 1610.01  670.29 1636.53  668.96
#Mann= 3 , 0 , 0
       0     .06       0  849.03     .04       0 1004.83      .1       0
Bank Sta=849.03,1004.83
XS Rating Curve= 0
Exp/Cntr=0.3,0.1

Type RM Length L Ch R = 1 ,119954.9,480.65,481.08,509.04
XS GIS Cut Line= 3
      1979886.12       298486.94      1980720.78       297963.81
      1981191.01       297581.75
#Sta/Elev= 30
       0  678.25       5  675.69      15  676.94      30  676.57      35  674.71
      50  672.73      90  653.11     125  637.93     160  631.01     235  629.02
     350  631.59     475  631.16     490  632.73     515   628.2     560  628.75
     610  625.92     670  629.03  683.62  628.65     705  625.86     850  626.79
  882.49  639.49    1215  662.06    1260  651.45    1295  658.32    1345  661.81
 1370.01  664.85    1465  682.58    1515  686.05    1545  685.15 1590.93  675.74
#Mann= 3 , 0 , 0
       0     .06       0  683.62     .04       0  882.49      .1       0
Bank Sta=683.62,882.49
XS Rating Curve= 0
Exp/Cntr=0.3,0.1

Type RM Length L Ch R = 1 ,119473.8,572.82,572.79,549.82
XS GIS Cut Line= 2
      1980238.79       298839.62      1981655.37       297910.91
#Sta/Elev= 30
       0  653.57   10.01   651.7   55.01  636.93     100  631.03     130  632.77
  225.01  630.18     355  629.36  415.01   630.6  440.01  627.39  480.01  629.81
  630.01  630.13     670  631.95  700.01  625.94  835.01  627.44     840  628.11
  850.01  635.71  855.01  637.38  867.77  638.35 1195.01  651.84 1250.01  655.74
 1270.01  659.22 1305.01  652.21 1485.01  665.35    1510  662.97 1530.01  662.81
    1615  668.85 1640.01   669.1 1655.01   670.8 1665.01  673.53 1693.87  667.55
#Mann= 3 , 0 , 0
       0     .06       0     670     .04       0  867.77      .1       0
Bank Sta=670,867.77
XS Rating Curve= 0
Exp/Cntr=0.3,0.1

Type RM Length L Ch R = 1 ,118901.0,657.47,600.49,606.85
XS GIS Cut Line= 3
      1980632.61       299262.82      1981373.23       298774.96
      1981925.75       298210.68
#Sta/Elev= 30
       0  657.74      95  653.07     155     644     210   631.4  395.01  627.39
     430  631.25     475  631.56     520  628.03     640  628.02     660  625.45
     835  626.26     880  630.67     910  631.57     945  628.51     975  628.79
     980  629.01  990.01  635.23    1015  636.37    1260  640.85    1295  639.73
    1345  643.11    1410  643.66    1415  643.86    1440  651.09    1470  647.08
    1505  648.94    1550  648.43 1605.01  661.72    1645  665.46  1676.6  662.87
#Mann= 3 , 0 , 0
       0     .06       0     640     .04       0     880      .1       0
Bank Sta=640,880
XS Rating Curve= 0
Exp/Cntr=0.3,0.1

Type RM Length L Ch R = 1 ,118300.5,520.94,546.6,459.51
XS GIS Cut Line= 3
      1981155.75       299697.79      1981843.46       299139.39
        1982369.         298471.
#Sta/Elev= 30
       0  670.18      20  670.61      45  679.62      85  675.85     140  675.47
     250  656.77     285  641.31     310  634.12     380  630.93     400  625.13
     460  626.22     610  622.94     675  625.44     795  625.18     855  622.56
  879.99  630.71    1000  632.05 1024.99  634.09    1045  633.46    1070  628.56
    1095  627.94    1105  633.38    1430  637.48    1460  639.67 1479.99   647.6
    1490  648.92    1550  640.71    1590  648.93    1615  643.85    1760     662
#Mann= 3 , 0 , 0
       0     .06       0     380     .04       0  879.99      .1       0
Bank Sta=380,879.99
XS Rating Curve= 0
Exp/Cntr=0.3,0.1

Type RM Length L Ch R = 1 ,117753.9,543.22,573.1,586.42
XS GIS Cut Line= 4
       1981499.6       300082.79      1982034.49        299653.7
      1982328.38       299271.64      1982698.69       298719.12
#Sta/Elev= 30
       0  728.39      65  739.41      70  741.05      90  753.42     145  747.66
     205  744.11     270  734.88     340  714.19     445  638.61  470.01  625.66
     580  622.47     885  623.16     890  623.32     910  630.62     915  630.95
    1125  629.58    1235   630.9    1260  629.07 1280.01  629.65    1295  632.32
    1575  633.24    1595  641.26    1610   645.8 1615.01  645.75    1655  635.35
    1660  635.49    1710  638.29    1750  646.26    1775  643.64 1832.89  654.57
#Mann= 3 , 0 , 0
       0     .06       0     445     .04       0 1615.01      .1       0
Bank Sta=445,1615.01
XS Rating Curve= 0
Exp/Cntr=0.3,0.1

Type RM Length L Ch R = 1 ,117180.8,782.54,779.51,923.5
XS GIS Cut Line= 3
      1981828.76       300511.88      1982551.74        299947.6
       1983174.8       299048.28
#Sta/Elev= 30
       0  725.33     130  741.48  240.01  727.49     320  704.47  410.01  666.81
     440  650.41  465.01  637.94  515.01  626.68     565   623.1     695  621.17
     850  622.33  875.01  631.09 1295.01  627.74    1490  630.51 1520.01  628.05
 1535.01  630.45 1550.01  628.72 1570.01  631.48 1765.01  634.49 1790.01  632.08
    1800  632.97 1825.01  645.76    1860  635.24 1885.01  636.27 1905.01   643.7
    1920  645.46 1945.01  640.15 1975.01  652.51 1985.01  659.03 2011.19  660.82
#Mann= 3 , 0 , 0
       0     .06       0     440     .04       0 1825.01      .1       0
Bank Sta=440,1825.01
XS Rating Curve= 0
Exp/Cntr=0.3,0.1

Type RM Length L Ch R = 1 ,116401.3,887.99,817.13,775.89
XS GIS Cut Line= 3
      1982316.63        301117.3      1983257.09       300364.93
        1984002.         299506.
#Sta/Elev= 30
       0  734.86      35  738.33      85  751.87     120  763.87     155  767.73
     275  735.98     335  718.06     440  666.28     465  657.36     525   630.3
     545  624.33     575  621.65     765  621.19     780  624.36    1015  627.97
    1510  625.82    1915   627.9    1945  628.84    1950  630.53    1965  643.01
 1974.64  644.17 1994.99   639.9    2020  628.74    2070  638.75 2100.01  630.58
    2195  635.33    2205  637.03    2230  645.89    2245  649.44    2363     662
#Mann= 3 , 0 , 0
       0     .06       0     465     .04       0 1974.64      .1       0
Bank Sta=465,1974.64
XS Rating Curve= 0
Exp/Cntr=0.3,0.1

Type RM Length L Ch R = 1 ,115584.2,671.15,684.36,731.47
XS GIS Cut Line= 2
      1982933.81       301763.87      1984603.13       300041.64
#Sta/Elev= 30
       0  720.63      95  725.68     105  719.27     110  718.31     145  720.16
     160  718.55     180  723.39     305  720.29     350  703.76     450  654.31
     470  643.81     495  635.36     515   621.8     575  621.68     660  621.84
     715  624.77     825   625.9    1425   625.6    1440  623.85 1470.01  625.95
    1840  627.12    1940   631.1    1995  643.83    2025  638.69    2085  642.21
    2110  647.83    2290  665.62    2330   678.6    2380  680.92 2398.48  675.35
#Mann= 3 , 0 , 0
       0     .06       0     450     .04       0    1995      .1       0
Bank Sta=450,1995
XS Rating Curve= 0
Exp/Cntr=0.3,0.1

Type RM Length L Ch R = 1 ,114899.8,901.83,914.18,1006.65
XS GIS Cut Line= 2
      1983409.92       302228.22      1985167.41       300523.63
#Sta/Elev= 30
       0  715.49      70  720.47      90  719.29     170  728.57     265  720.51
     350  716.27  364.99  709.95     465  650.75     480  640.62     515  623.08
     520  622.01     665  621.46     680  625.11     735  625.51 1284.99  623.88
    1620  625.61    1675  627.37    1705  625.82    1755   628.4    1820  628.33
    1900  632.67    1920   636.4 1980.71  642.36    1990  643.08    2010  640.03
    2035  638.59 2099.99  640.04 2279.99  648.52    2400  663.21 2448.35  661.61
#Mann= 3 , 0 , 0
       0     .06       0     465     .04       0 1980.71      .1       0
Bank Sta=465,1980.71
XS Rating Curve= 0
Exp/Cntr=0.3,0.1

Type RM Length L Ch R = 1 ,113985.6,1115.1,1128.67,1236.81
XS GIS Cut Line= 2
      1983983.01       302918.87       1985952.1       301108.48
#Sta/Elev= 30
       0  700.02     155  711.29     405  705.24     435  702.52     480  680.15
     505   664.4     525  649.03     540  638.51  570.01  621.33     720   621.3
     725   622.8     735  623.49    1335  623.42    1535  621.58    1570   623.3
    1625  623.67    1665  626.92    1690  625.71    1740  628.78    1755  632.56
    1860  640.52    2070  641.57 2110.01  639.94    2145  644.84 2163.42  644.99
    2205   643.4    2405  648.52    2585  660.58    2620  664.94 2674.85  666.13
#Mann= 3 , 0 , 0
       0     .06       0     525     .04       0 2163.42      .1       0
Bank Sta=525,2163.42
XS Rating Curve= 0
Exp/Cntr=0.3,0.1

Type RM Length L Ch R = 1 ,112856.9,967.42,885.95,879.35
XS GIS Cut Line= 2
      1984888.21       303536.05      1986951.34       301878.48
#Sta/Elev= 30
       0  671.47      20  675.47      55  686.83      80  690.11     135  702.42
  194.99   696.8     225  695.88     320  687.17  354.99  679.32     385  669.53
  439.99  640.31  464.99  626.61     495   621.3     775  622.37 1249.99  621.18
    1545  621.38    1590  623.81 1664.99  632.66    1810  634.85    1840  639.93
    1875  635.44    1890  635.31 1924.99  638.59 1989.99  637.14 2289.99  645.49
    2515  657.45 2564.99  667.98    2610  674.31    2620  674.58 2646.52  669.39
#Mann= 3 , 0 , 0
       0     .06       0  439.99     .04       0    1840      .1       0
Bank Sta=439.99,1840
XS Rating Curve= 0
Exp/Cntr=0.3,0.1

Type RM Length L Ch R = 1 ,111971.0,1123.83,1313.57,1116.57
XS GIS Cut Line= 3
      1985537.71       304273.72      1986460.54       303227.46
      1987630.24       302475.09
#Sta/Elev= 30
       0  676.02      70  679.83     180  682.52  304.99  667.91     340  666.45
     385  652.34     415  638.37     450   621.3     760   621.3     780  622.37
    1150   621.3    1220  622.43 1634.99   621.3    1650  623.67    1700  623.24
    1735   624.2    1830  630.27    1900  630.15    1930  635.58    1940  635.46
    1965  632.01    2100  633.54    2195  636.33 2249.99   639.5    2425  645.68
 2614.99  654.56    2700  659.58    2750  663.33    2770  666.63 2785.87  666.75
#Mann= 3 , 0 , 0
       0     .06       0     415     .04       0    1930      .1       0
Bank Sta=415,1930
XS Rating Curve= 0
Exp/Cntr=0.3,0.1

Type RM Length L Ch R = 1 ,110657.4,1070.91,997.52,929.31
XS GIS Cut Line= 2
      1986342.98       305031.97      1988476.66       303098.15
#Sta/Elev= 30
       0  676.38      85   677.7     215  676.05     240  672.17     265  671.22
     300  673.54     360  675.23     455   664.5     530  658.44     555  650.12
     605  622.96  610.01  621.17     650  618.37     780  613.12  850.01  618.84
    1190  620.61    1590  619.85    1650   621.7    1690  626.17    1715   631.9
    1740  630.31    1775  624.24 1845.01  626.34    2480  636.36    2560  639.58
    2620  643.45    2705  653.45    2870  668.51    2875  668.49 2879.63  666.67
#Mann= 3 , 0 , 0
       0     .06       0     555     .04       0    1715      .1       0
Bank Sta=555,1715
XS Rating Curve= 0
Exp/Cntr=0.3,0.1

Type RM Length L Ch R = 1 ,109659.9,1058.87,1059.82,1098.85
XS GIS Cut Line= 3
      1987160.01       305713.81      1987724.29        305131.9
        1989170.         303638.
#Sta/Elev= 30
       0  670.74     120   670.2     180   667.7     225  668.02     280  673.45
     335   675.3     395  667.42     480  662.75     545  655.98  665.01  636.69
     750     620  810.57  616.05     830  615.93     860  618.87     990  616.86
    1370  619.06    1410  617.03    1530  621.57    1570  633.46    1575  633.87
    1585  633.93 1590.01  632.57    1600  626.69    1615  622.78 1660.01  624.49
    1690  621.33    2300  628.72    2465  633.75 2797.56  649.18    2907     662
#Mann= 3 , 0 , 0
       0     .06       0  665.01     .04       0    1575      .1       0
Bank Sta=665.01,1575
XS Rating Curve= 0
Exp/Cntr=0.3,0.1

Type RM Length L Ch R = 1 ,108600.1,1299.23,1266.45,1255.15
XS GIS Cut Line= 2
      1988009.36       306292.78        1990080.         304330.
#Sta/Elev= 30
       0  671.88      90   673.1     115  669.71     125  672.11     130  676.92
     220  674.59     320  663.39     360  657.09     420  641.79     460  634.28
  520.01  623.53     570  619.67     770  615.96     820  611.97     910  609.49
     930  610.16  975.01  617.73 1095.01  617.77    1150  616.33    1275  621.25
    1295  626.56 1320.01  629.01    1360   621.3 1770.01  621.36 2335.01  630.57
 2450.01   633.5    2595  640.41 2630.01  634.77 2755.01  647.71    2850     662
#Mann= 3 , 0 , 0
       0     .06       0     460     .04       0 1320.01      .1       0
Bank Sta=460,1320.01
XS Rating Curve= 0
Exp/Cntr=0.3,0.1

Type RM Length L Ch R = 1 ,107333.6,826.39,867.68,932.05
XS GIS Cut Line= 2
      1988949.83       307174.46       1991083.5       305076.06
#Sta/Elev= 30
       0  674.91   14.99  675.07   89.99  667.46     155  665.02     195  661.11
  239.99  651.22     265  647.14  384.99  632.54  409.99   631.6     465  621.27
     575  619.79     770  612.67     825  616.27  904.99  616.12    1185  622.88
    1260  620.58    1480   617.4    1620  617.05    1795  618.31    1835  620.85
    1860  619.26    2225  621.95 2549.99  635.97    2640  635.23    2700  636.36
    2895  652.29    2955  658.74    2965  658.41    2975  661.79 2992.63   662.7
#Mann= 3 , 0 , 0
       0     .06       0  384.99     .04       0    1185      .1       0
Bank Sta=384.99,1185
XS Rating Curve= 0
Exp/Cntr=0.3,0.1

Type RM Length L Ch R = 1 ,106466.0,1160.36,1287.33,1476.96
XS GIS Cut Line= 2
      1989481.78       307782.82      1991856.44       305737.32
#Sta/Elev= 30
       0  674.15     175  667.14     235  667.41     280  664.72  294.99  659.98
  379.99  622.33  399.99  613.09     470  609.48     570  611.41  609.99   616.7
  994.99  615.46 1094.99  616.67 1159.99  621.46    1200  622.91 1239.99  620.07
    1280  619.83 1299.99  617.22 1409.99  615.66 1519.99  617.62 1749.99  617.69
 2164.99  620.67 2589.99  628.25    2635  628.45    2665  626.95 2689.99  630.36
    2775  633.25 3009.99  647.15 3079.99  653.32 3124.99   659.3 3134.18  664.24
#Mann= 3 , 0 , 0
       0     .06       0  379.99     .04       0    1200      .1       0
Bank Sta=379.99,1200
XS Rating Curve= 0
Exp/Cntr=0.3,0.1
